--- StephenvilleCrossi.prj (project) ---

Proj Title=Stephenville Crossing Model
Current Plan=p28
Default Exp/Contr=0.3,0.1
SI Units
Geom File=g11
Flow File=f01
Flow File=f02
Flow File=f03
Unsteady File=u05
Unsteady File=u06
Unsteady File=u08
Unsteady File=u09
Unsteady File=u18
Unsteady File=u22
Unsteady File=u23
Unsteady File=u24
Unsteady File=u25
Unsteady File=u26
Unsteady File=u27
Unsteady File=u28
Unsteady File=u29
Unsteady File=u30
Unsteady File=u31
Unsteady File=u32
Unsteady File=u33
Unsteady File=u34
Unsteady File=u35
Unsteady File=u36
Unsteady File=u37
Plan File=p07
Plan File=p08
Plan File=p10
Plan File=p11
Plan File=p24
Plan File=p25
Plan File=p26
Plan File=p27
Plan File=p28
Plan File=p29
Plan File=p30
Plan File=p31
Plan File=p32
Plan File=p33
Plan File=p34
Plan File=p35
Plan File=p36
Plan File=p37
Plan File=p38
Plan File=p39
Plan File=p40
Plan File=p41
Y Axis Title=Elevation
X Axis Title(PF)=Main Channel Distance
X Axis Title(XS)=Station
BEGIN DESCRIPTION:
END DESCRIPTION:
DSS File=dss
DSS Export Rating Curves= 0
DSS Export Rating Curve Sorted= 0
DSS Export Volume Flow Curves= 0
DXF OffsetX= 0
DXF OffsetY= 0
DXF ScaleX= 1
DXF ScaleY= 10

--- StephenvilleCrossi.p28 (plan) ---

Plan Title=100yr,HighTide,-2hrOffset_CRITICAL
Program Version=4.10
Short Identifier=100yr,high,-2hr
Simulation Date=07Jun1995,0000,10JUN1995,2300
Geom File=g11
Flow File=u25
Mixed Flow
K Sum by GR= 0
Std Step Tol= 0.003
Critical Tol= 0.003
Num of Std Step Trials= 20
Max Error Tol= 0.1
Flow Tol Ratio= 0.001
Split Flow NTrial= 30
Split Flow Tol= 0.006
Split Flow Ratio= 0.02
Log Output Level= 0
Friction Slope Method= 1
Unsteady Friction Slope Method= 2
Unsteady Bridges Friction Slope Method= 1
Parabolic Critical Depth
Global Vel Dist= 0 , 0 , 0
Global Log Level= 0
CheckData=True
Encroach Param=-1 ,0,0, 0
Computation Interval=1MIN
Output Interval=1HOUR
Run HTab= 1
Run UNet= 1
Run PostProcess= 1
Run WQNet= 0
UNET Theta= 0.6
UNET Theta Warmup= 1
UNET ZTol= 0.006
UNET ZSATol= 0.015
UNET MxIter= 20
UNET MaxInSteps= 0
UNET DtIC= 0
UNET DtMin= 0
UNET MaxCRTS= 20
UNET WFStab= 2
UNET SFStab= 1
UNET WFX= 1
UNET SFX= 1
UNET DSS MLevel= 4
UNET DZMax Abort= 30
UNET Convert EG Bridges= 0
UNET Use Existing IB Tables=-1
UNET Froude Reduction=False
UNET Froude Limit= 1
UNET Froude Power= 10
UNET Time Slicing=0,0, 5
UNET Junction Losses=0
Instantaneous Interval=1HOUR
DSS File=dss
Write IC File= 0
Write IC File at Sim End=0
Echo Input=False
Echo Parameters=False
Echo Output=False
Write Detailed= 0
WQ AD Non Conservative
WQ ULTIMATE=-1
WQ Max Comp Step=1HOUR
WQ Output Interval=15MIN
WQ Output Selected Increments= 0
WQ Output face flow=0
WQ Output face velocity=0
WQ Output face area=0
WQ Output face dispersion=0
WQ Output cell volume=0
WQ Output cell surface area=0
WQ Output cell continuity=0
WQ Output cumulative cell continuity=0
WQ Output face conc=0
WQ Output face dconc_dx=0
WQ Output face courant=0
WQ Output face peclet=0
WQ Output face adv mass=0
WQ Output face disp mass=0
WQ Output cell mass=0
WQ Output cell source sink temp=0
WQ Output cell source sink nsm=0
WQ Output MaxMinRange=-1
WQ Daily Max Min Mean=-1
WQ Daily Range=0
WQ Daily Time=0
WQ Create Restart=0
WQ Fixed Restart=0
WQ System Summary=0
WQ Use Fixed Temperature=0
Sorting and Armoring Iterations= 10
XS Update Threshold= 0.02
Hydraulics Update Threshold= 0.02
Energy Slope Method= 1
Volume Change Method= 0
XS Weighting Method= 0
Number of US Weighted Cross Sections= 1
Number of DS Weighted Cross Sections= 1
Upstream XS Weight=0.25
Main XS Weight=0.5
Downstream XS Weight=0.25
Number of DS XS's Weighted with US Boundary= 1
Upstream Boundary Weight= 1
Weight of XSs Associated with US Boundary= 0
Number of US XS's Weighted with DS Boundary= 1
Downstream Boundary Weight= 0.5
Weight of XSs Associated with DS Boundary= 0.5
Sediment Output Level= 4
Mass or Volume Output= 0
Output Increment Type= 1
Profile and TS Output Increment= 10
XS Output Flag= 0
XS Output Increment= 10
Disregard all LS=0
Disregard all Conn=0
Disregard all Breaches=0
Disregard all Pumps=0

--- StephenvilleCrossi.p01 (plan) ---

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Plan Title=Plan 01
Short Identifier=Plan 01
Geom File=g01
Flow File=f01
Subcritical Flow
Computation Interval=1HOUR
Run HTab= 0
Run UNet= 0
Run PostProcess= 0
UNET Theta= 1

--- StephenvilleCrossi.p07 (plan) ---

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Plan Title=100yr,HighTide,2hrOffset
Short Identifier=100,High,2hr
Geom File=g11
Flow File=u05

--- StephenvilleCrossi.p08 (plan) ---

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Plan Title=100yr,HighTide,1hrOffset
Short Identifier=100yr,High,1hr
Geom File=g11
Flow File=u06

--- StephenvilleCrossi.p10 (plan) ---

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Plan Title=100yr,HighTide,0hrOffset
Short Identifier=100yr,High,0hr
Geom File=g11
Flow File=u08

--- StephenvilleCrossi.p11 (plan) ---

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Plan Title=100yr,HighTide,3hrOffset
Short Identifier=100yr.high,3hr
Geom File=g11
Flow File=u09

--- StephenvilleCrossi.p24 (plan) ---

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Plan Title=Calib_1986_Mar9,11
Short Identifier=Calib1986_Mar9
Simulation Date=2DEC1986,16:00,20DEC1986,11:00
Geom File=g11
Flow File=u18
Subcritical Flow

--- StephenvilleCrossi.p25 (plan) ---

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Plan Title=Calibration-highwater-Nov2010,Mar10,11
Short Identifier=CalibHigh,Mar10
Simulation Date=03NOV2010,2000,07NOV2010,1600
Geom File=g11
Flow File=u22

--- StephenvilleCrossi.p26 (plan) ---

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Plan Title=Calibration-surveydate-Sep2010,Mar10,11
Short Identifier=Calib_Surv_Mar10
Simulation Date=25SEP2010,0000,28SEP2010,2300
Geom File=g11
Flow File=u23

--- StephenvilleCrossi.p27 (plan) ---

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Plan Title=100yr,HighTide,-1hrOffset
Short Identifier=100,high,-1
Geom File=g11
Flow File=u24

--- StephenvilleCrossi.p29 (plan) ---

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Plan Title=100yr,HighTide,-3hrOffset
Short Identifier=100yr,high,-3hr
Geom File=g11
Flow File=u26

--- StephenvilleCrossi.p30 (plan) ---

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Plan Title=100yr,HighTide,-4hrOffset
Short Identifier=100yr,high,-4hr
Geom File=g11
Flow File=u27

--- StephenvilleCrossi.f01 (steady flow) ---

Flow Title=Steady State Test
Program Version=4.10
Number of Profiles= 2
Profile Names=1:20,1:100
River Rch & RM=Harrys River,Upstream        ,1826.936
     648     822
River Rch & RM=Main Gut,Downstream      ,486.6117
    2054    2604
River Rch & RM=StGeorgesRiver,Upstream        ,3118.381
    1406    1782
Boundary for River Rch & Prof#=Harrys River,Upstream        , 1
Up Type= 2
Dn Type= 0
Boundary for River Rch & Prof#=Harrys River,Upstream        , 2
Up Type= 2
Dn Type= 0
Boundary for River Rch & Prof#=Main Gut,Downstream      , 1
Up Type= 0
Dn Type= 1
Dn Known WS=0
Boundary for River Rch & Prof#=Main Gut,Downstream      , 2
Up Type= 0
Dn Type= 1
Dn Known WS=0
Boundary for River Rch & Prof#=StGeorgesRiver,Upstream        , 1
Up Type= 2
Dn Type= 0
Boundary for River Rch & Prof#=StGeorgesRiver,Upstream        , 2
Up Type= 2
Dn Type= 0
DSS Import GetInterval= 0
DSS Import GetPeak= 0
DSS Import FillOption= 0
Storage Area Elev=13              , 2
       0       0

--- StephenvilleCrossi.f02 (steady flow) ---

Flow Title=ExtremeTide,NormalFlow
Program Version=4.10
Number of Profiles= 2
Profile Names=1:20,1:100
River Rch & RM=Harrys River,Upstream        ,1826.936
    22.2    22.2
River Rch & RM=Main Gut,Downstream      ,600
    43.8    43.8
River Rch & RM=StGeorgesRiver,Upstream        ,1500
      66      66
Boundary for River Rch & Prof#=Harrys River,Upstream        , 1
Up Type= 2
Dn Type= 0
Boundary for River Rch & Prof#=Harrys River,Upstream        , 2
Up Type= 2
Dn Type= 0
Boundary for River Rch & Prof#=Main Gut,Downstream      , 1
Up Type= 0
Dn Type= 1
Dn Known WS=1.2
Boundary for River Rch & Prof#=Main Gut,Downstream      , 2
Up Type= 0
Dn Type= 1
Dn Known WS=1.4
Boundary for River Rch & Prof#=StGeorgesRiver,Upstream        , 1
Up Type= 2
Dn Type= 0
Boundary for River Rch & Prof#=StGeorgesRiver,Upstream        , 2
Up Type= 2
Dn Type= 0
DSS Import GetInterval= 0
DSS Import GetPeak= 0
DSS Import FillOption= 0
Storage Area Elev=St. George's Riv, 2
     1.2     1.4

--- StephenvilleCrossi.f03 (steady flow) ---

Flow Title=Flow 03
Program Version=4.10
Number of Profiles= 1
Profile Names=PF 1
DSS Import GetInterval= 0
DSS Import GetPeak= 0
DSS Import FillOption= 0

--- StephenvilleCrossi.u25 (unsteady flow) ---

Flow Title=1:100, High Tide, -2hr offset
Program Version=4.10
Use Restart= 0
Initial Flow Loc=Harrys River    ,Upstream        ,1826.936,51.3
Initial Flow Loc=Main Gut        ,Downstream      ,600     ,152.6
Initial Flow Loc=StGeorgesRiver  ,Upstream        ,1500    ,101.3
Initial Storage Elev=St. George's Riv,0.358
Boundary Location=Harrys River    ,Upstream        ,1826.936,        ,                ,                ,
Interval=1HOUR
Flow Hydrograph= 96
    51.3    51.2    51.1      51    50.9    50.9    50.8    50.7    50.6    50.5
    50.4    50.3    50.1      50    49.9    49.7    49.5    49.3    49.1    48.8
    48.6    48.4    48.1    48.2    48.3    48.4    48.4    49.4    49.9    50.2
    51.7    55.8    93.3   162.9   262.3   372.8   829.9   888.2   946.8   934.8
   844.8   782.5   724.7   668.3   612.6     613   612.3   611.4   610.4   621.5
   633.1   639.7   607.2   575.7   543.5   509.8     476   442.3   410.6   375.4
   354.7   335.8     319   306.1   292.4   280.8   267.1   257.9   251.5     245
   238.6   232.2     225   217.3   214.1   211.7   209.3   206.5   204.1   201.7
   199.2     197   194.6   192.2   189.8   187.5   185.2   182.8   180.4   178.4
     176   173.5   171.5   169.5   167.6   165.9
Use DSS=False
CWMS InputPosition= 0
Use Fixed Start Time=False
Fixed Start Date/Time=07JUN1995,0000
Is Critical Boundary=False
Boundary Location=StGeorgesRiver  ,Upstream        ,1500    ,        ,                ,                ,
Interval=1HOUR
Flow Hydrograph= 96
   101.3   101.1   100.9   100.8   100.6   100.5   100.3   100.2    99.9    99.7
    99.5    99.3      99    98.8    98.6    98.3    97.8    97.3      97    96.3
      96    95.7    95.1    95.2    95.4    95.6    95.7    97.6    98.6    99.2
   102.2   110.2   184.4   321.7   518.2   736.5  1639.6  1754.7  1870.6  1846.8
    1669    1546  1431.7  1320.2  1210.3  1211.1  1209.7  1207.9    1206  1227.8
  1250.8  1263.9  1199.6  1137.3  1073.8  1007.1   940.5   873.8   811.1   741.7
   700.8   663.5   630.1   604.7   577.8   554.7   527.8   509.5   496.8   484.1
   471.4   458.7   444.5   429.4     423   418.2   413.5   407.9   403.2   398.4
   393.4   389.3   384.5   379.8     375   370.4   365.9   361.1   356.3   352.4
   347.6   342.8   338.8   334.8     331   327.7
Use DSS=False
CWMS InputPosition= 0
Use Fixed Start Time=False
Fixed Start Date/Time=07JUN1995,0000
Is Critical Boundary=False
Boundary Location=Main Gut        ,Downstream      ,0       ,        ,                ,                ,
Interval=1HOUR
Stage Hydrograph= 96
    .358     .27    .073   -.187   -.451   -.659   -.759   -.716   -.534   -.257
    .052    .322    .478    .483    .346    .113   -.154    -.39   -.542    -.57
   -.458   -.239    .024    .264    .417    .431    .298    .051   -.243   -.512
     -.7   -.766   -.678    -.45   -.151    .145    .373    .475     .42    .224
    -.05    -.32   -.527   -.632   -.596   -.413   -.141    .141    .371    .495
     .47     .29    .008   -.293    -.54   -.695   -.718   -.585   -.331   -.042
    .212    .385    .426    .309    .066   -.221   -.468    -.63   -.677   -.574
   -.335   -.037    .237    .441    .532    .469    .256   -.035   -.314   -.524
   -.637   -.619   -.455   -.206    .043    .241    .353    .334    .167   -.098
   -.369   -.576   -.687   -.676   -.519   -.251
Use DSS=False
CWMS InputPosition= 0
Use Fixed Start Time=False
Fixed Start Date/Time=07JUN1995,0000
Is Critical Boundary=False

--- StephenvilleCrossi.u05 (unsteady flow) ---

Flow Title=1:100, High Tide, 2hr offset
Program Version=4.10
Use Restart= 0
Initial Flow Loc=Harrys River    ,Upstream        ,1826.936,51.3
Initial Flow Loc=Main Gut        ,Downstream      ,600     ,152.6
Initial Flow Loc=StGeorgesRiver  ,Upstream        ,1500    ,101.3
Initial Storage Elev=St. George's Riv,-0.085
Boundary Location=Harrys River    ,Upstream        ,1826.936,        ,                ,                ,
Interval=1HOUR
Flow Hydrograph= 96
    51.3    51.2    51.1      51    50.9    50.9    50.8    50.7    50.6    50.5
    50.4    50.3    50.1      50    49.9    49.7    49.5    49.3    49.1    48.8
    48.6    48.4    48.1    48.2    48.3    48.4    48.4    49.4    49.9    50.2
    51.7    55.8    93.3   162.9   262.3   372.8   829.9   888.2   946.8   934.8
   844.8   782.5   724.7   668.3   612.6     613   612.3   611.4   610.4   621.5
   633.1   639.7   607.2   575.7   543.5   509.8     476   442.3   410.6   375.4
   354.7   335.8     319   306.1   292.4   280.8   267.1   257.9   251.5     245
   238.6   232.2     225   217.3   214.1   211.7   209.3   206.5   204.1   201.7
   199.2     197   194.6   192.2   189.8   187.5   185.2   182.8   180.4   178.4
     176   173.5   171.5   169.5   167.6   165.9
Use DSS=False
CWMS InputPosition= 0
Use Fixed Start Time=True
Fixed Start Date/Time=07JUN1995,0000
Is Critical Boundary=False
Boundary Location=StGeorgesRiver  ,Upstream        ,1500    ,        ,                ,                ,
Interval=1HOUR
Flow Hydrograph= 96
   101.3   101.1   100.9   100.8   100.6   100.5   100.3   100.2    99.9    99.7
    99.5    99.3      99    98.8    98.6    98.3    97.8    97.3      97    96.3
      96    95.7    95.1    95.2    95.4    95.6    95.7    97.6    98.6    99.2
   102.2   110.2   184.4   321.7   518.2   736.5  1639.6  1754.7  1870.6  1846.8
    1669    1546  1431.7  1320.2  1210.3  1211.1  1209.7  1207.9    1206  1227.8
  1250.8  1263.9  1199.6  1137.3  1073.8  1007.1   940.5   873.8   811.1   741.7
   700.8   663.5   630.1   604.7   577.8   554.7   527.8   509.5   496.8   484.1
   471.4   458.7   444.5   429.4     423   418.2   413.5   407.9   403.2   398.4
   393.4   389.3   384.5   379.8     375   370.4   365.9   361.1   356.3   352.4
   347.6   342.8   338.8   334.8     331   327.7
Use DSS=False
CWMS InputPosition= 0
Use Fixed Start Time=True
Fixed Start Date/Time=07JUN1995,0000
Is Critical Boundary=False
Boundary Location=Main Gut        ,Downstream      ,0       ,        ,                ,                ,
Interval=1HOUR
Stage Hydrograph= 96
   -.085    .143    .311    .358     .27    .073   -.187   -.451   -.659   -.759
   -.716   -.534   -.257    .052    .322    .478    .483    .346    .113   -.154
    -.39   -.542    -.57   -.458   -.239    .024    .264    .417    .431    .298
    .051   -.243   -.512     -.7   -.766   -.678    -.45   -.151    .145    .373
    .475     .42    .224    -.05    -.32   -.527   -.632   -.596   -.413   -.141
    .141    .371    .495     .47     .29    .008   -.293    -.54   -.695   -.718
   -.585   -.331   -.042    .212    .385    .426    .309    .066   -.221   -.468
    -.63   -.677   -.574   -.335   -.037    .237    .441    .532    .469    .256
   -.035   -.314   -.524   -.637   -.619   -.455   -.206    .043    .241    .353
    .334    .167   -.098   -.369   -.576   -.687
Use DSS=False
CWMS InputPosition= 0
Use Fixed Start Time=True
Fixed Start Date/Time=07JUN1995,0000
Is Critical Boundary=False

--- StephenvilleCrossi.u06 (unsteady flow) ---

Flow Title=1:100, High Tide, 1hr offset
Program Version=4.10
Use Restart= 0
Initial Flow Loc=Harrys River    ,Upstream        ,1826.936,51.3
Initial Flow Loc=Main Gut        ,Downstream      ,600     ,152.6
Initial Flow Loc=StGeorgesRiver  ,Upstream        ,1500    ,101.3
Initial Storage Elev=St. George's Riv,0.143
Boundary Location=Harrys River    ,Upstream        ,1826.936,        ,                ,                ,
Interval=1HOUR
Flow Hydrograph= 96
    51.3    51.2    51.1      51    50.9    50.9    50.8    50.7    50.6    50.5
    50.4    50.3    50.1      50    49.9    49.7    49.5    49.3    49.1    48.8
    48.6    48.4    48.1    48.2    48.3    48.4    48.4    49.4    49.9    50.2
    51.7    55.8    93.3   162.9   262.3   372.8   829.9   888.2   946.8   934.8
   844.8   782.5   724.7   668.3   612.6     613   612.3   611.4   610.4   621.5
   633.1   639.7   607.2   575.7   543.5   509.8     476   442.3   410.6   375.4
   354.7   335.8     319   306.1   292.4   280.8   267.1   257.9   251.5     245
   238.6   232.2     225   217.3   214.1   211.7   209.3   206.5   204.1   201.7
   199.2     197   194.6   192.2   189.8   187.5   185.2   182.8   180.4   178.4
     176   173.5   171.5   169.5   167.6   165.9
Use DSS=False
CWMS InputPosition= 0
Use Fixed Start Time=True
Fixed Start Date/Time=07JUN1995,0000
Is Critical Boundary=False
Boundary Location=StGeorgesRiver  ,Upstream        ,1500    ,        ,                ,                ,
Interval=1HOUR
Flow Hydrograph= 96
   101.3   101.1   100.9   100.8   100.6   100.5   100.3   100.2    99.9    99.7
    99.5    99.3      99    98.8    98.6    98.3    97.8    97.3      97    96.3
      96    95.7    95.1    95.2    95.4    95.6    95.7    97.6    98.6    99.2
   102.2   110.2   184.4   321.7   518.2   736.5  1639.6  1754.7  1870.6  1846.8
    1669    1546  1431.7  1320.2  1210.3  1211.1  1209.7  1207.9    1206  1227.8
  1250.8  1263.9  1199.6  1137.3  1073.8  1007.1   940.5   873.8   811.1   741.7
   700.8   663.5   630.1   604.7   577.8   554.7   527.8   509.5   496.8   484.1
   471.4   458.7   444.5   429.4     423   418.2   413.5   407.9   403.2   398.4
   393.4   389.3   384.5   379.8     375   370.4   365.9   361.1   356.3   352.4
   347.6   342.8   338.8   334.8     331   327.7
Use DSS=False
CWMS InputPosition= 0
Use Fixed Start Time=True
Fixed Start Date/Time=07JUN1995,0000
Is Critical Boundary=False
Boundary Location=Main Gut        ,Downstream      ,0       ,        ,                ,                ,
Interval=1HOUR
Stage Hydrograph= 96
    .143    .311    .358     .27    .073   -.187   -.451   -.659   -.759   -.716
   -.534   -.257    .052    .322    .478    .483    .346    .113   -.154    -.39
   -.542    -.57   -.458   -.239    .024    .264    .417    .431    .298    .051
   -.243   -.512     -.7   -.766   -.678    -.45   -.151    .145    .373    .475
     .42    .224    -.05    -.32   -.527   -.632   -.596   -.413   -.141    .141
    .371    .495     .47     .29    .008   -.293    -.54   -.695   -.718   -.585
   -.331   -.042    .212    .385    .426    .309    .066   -.221   -.468    -.63
   -.677   -.574   -.335   -.037    .237    .441    .532    .469    .256   -.035
   -.314   -.524   -.637   -.619   -.455   -.206    .043    .241    .353    .334
    .167   -.098   -.369   -.576   -.687   -.676
Use DSS=False
CWMS InputPosition= 0
Use Fixed Start Time=True
Fixed Start Date/Time=07JUN1995,0000
Is Critical Boundary=False

--- StephenvilleCrossi.u08 (unsteady flow) ---

Flow Title=1:100, High Tide, 0hr offset
Program Version=4.10
Use Restart= 0
Initial Flow Loc=Harrys River    ,Upstream        ,1826.936,51.3
Initial Flow Loc=Main Gut        ,Downstream      ,600     ,152.6
Initial Flow Loc=StGeorgesRiver  ,Upstream        ,1500    ,101.3
Initial Storage Elev=St. George's Riv,-0.574
Boundary Location=Harrys River    ,Upstream        ,1826.936,        ,                ,                ,
Interval=1HOUR
Flow Hydrograph= 96
    51.3    51.2    51.1      51    50.9    50.9    50.8    50.7    50.6    50.5
    50.4    50.3    50.1      50    49.9    49.7    49.5    49.3    49.1    48.8
    48.6    48.4    48.1    48.2    48.3    48.4    48.4    49.4    49.9    50.2
    51.7    55.8    93.3   162.9   262.3   372.8   829.9   888.2   946.8   934.8
   844.8   782.5   724.7   668.3   612.6     613   612.3   611.4   610.4   621.5
   633.1   639.7   607.2   575.7   543.5   509.8     476   442.3   410.6   375.4
   354.7   335.8     319   306.1   292.4   280.8   267.1   257.9   251.5     245
   238.6   232.2     225   217.3   214.1   211.7   209.3   206.5   204.1   201.7
   199.2     197   194.6   192.2   189.8   187.5   185.2   182.8   180.4   178.4
     176   173.5   171.5   169.5   167.6   165.9
Use DSS=False
CWMS InputPosition= 0
Use Fixed Start Time=False
Fixed Start Date/Time=07JUN1995,0000
Is Critical Boundary=False
Boundary Location=StGeorgesRiver  ,Upstream        ,1500    ,        ,                ,                ,
Interval=1HOUR
Flow Hydrograph= 96
   101.3   101.1   100.9   100.8   100.6   100.5   100.3   100.2    99.9    99.7
    99.5    99.3      99    98.8    98.6    98.3    97.8    97.3      97    96.3
      96    95.7    95.1    95.2    95.4    95.6    95.7    97.6    98.6    99.2
   102.2   110.2   184.4   321.7   518.2   736.5  1639.6  1754.7  1870.6  1846.8
    1669    1546  1431.7  1320.2  1210.3  1211.1  1209.7  1207.9    1206  1227.8
  1250.8  1263.9  1199.6  1137.3  1073.8  1007.1   940.5   873.8   811.1   741.7
   700.8   663.5   630.1   604.7   577.8   554.7   527.8   509.5   496.8   484.1
   471.4   458.7   444.5   429.4     423   418.2   413.5   407.9   403.2   398.4
   393.4   389.3   384.5   379.8     375   370.4   365.9   361.1   356.3   352.4
   347.6   342.8   338.8   334.8     331   327.7
Use DSS=False
CWMS InputPosition= 0
Use Fixed Start Time=False
Fixed Start Date/Time=07JUN1995,0000
Is Critical Boundary=False
Boundary Location=Main Gut        ,Downstream      ,0       ,        ,                ,                ,
Interval=1HOUR
Stage Hydrograph= 26
   -.574   -.335   -.037    .237    .441    .532    .469    .256   -.035   -.314
   -.524   -.637   -.619   -.455   -.206    .043    .241    .353    .334    .167
   -.098   -.369   -.576   -.687   -.676   -.519
Use DSS=False
CWMS InputPosition= 0
Use Fixed Start Time=False
Fixed Start Date/Time=07JUN1995,0000
Is Critical Boundary=False

--- StephenvilleCrossi.u09 (unsteady flow) ---

Flow Title=1:100, High Tide, 3hr offset
Program Version=4.10
Use Restart= 0
Initial Flow Loc=Harrys River    ,Upstream        ,1826.936,51.3
Initial Flow Loc=Main Gut        ,Downstream      ,600     ,152.6
Initial Flow Loc=StGeorgesRiver  ,Upstream        ,1500    ,101.3
Initial Storage Elev=St. George's Riv,0.311
Boundary Location=Harrys River    ,Upstream        ,1826.936,        ,                ,                ,
Interval=1HOUR
Flow Hydrograph= 96
    51.3    51.2    51.1      51    50.9    50.9    50.8    50.7    50.6    50.5
    50.4    50.3    50.1      50    49.9    49.7    49.5    49.3    49.1    48.8
    48.6    48.4    48.1    48.2    48.3    48.4    48.4    49.4    49.9    50.2
    51.7    55.8    93.3   162.9   262.3   372.8   829.9   888.2   946.8   934.8
   844.8   782.5   724.7   668.3   612.6     613   612.3   611.4   610.4   621.5
   633.1   639.7   607.2   575.7   543.5   509.8     476   442.3   410.6   375.4
   354.7   335.8     319   306.1   292.4   280.8   267.1   257.9   251.5     245
   238.6   232.2     225   217.3   214.1   211.7   209.3   206.5   204.1   201.7
   199.2     197   194.6   192.2   189.8   187.5   185.2   182.8   180.4   178.4
     176   173.5   171.5   169.5   167.6   165.9
Use DSS=False
CWMS InputPosition= 0
Use Fixed Start Time=False
Fixed Start Date/Time=07JUN1995,0000
Is Critical Boundary=False
Boundary Location=StGeorgesRiver  ,Upstream        ,1500    ,        ,                ,                ,
Interval=1HOUR
Flow Hydrograph= 96
   101.3   101.1   100.9   100.8   100.6   100.5   100.3   100.2    99.9    99.7
    99.5    99.3      99    98.8    98.6    98.3    97.8    97.3      97    96.3
      96    95.7    95.1    95.2    95.4    95.6    95.7    97.6    98.6    99.2
   102.2   110.2   184.4   321.7   518.2   736.5  1639.6  1754.7  1870.6  1846.8
    1669    1546  1431.7  1320.2  1210.3  1211.1  1209.7  1207.9    1206  1227.8
  1250.8  1263.9  1199.6  1137.3  1073.8  1007.1   940.5   873.8   811.1   741.7
   700.8   663.5   630.1   604.7   577.8   554.7   527.8   509.5   496.8   484.1
   471.4   458.7   444.5   429.4     423   418.2   413.5   407.9   403.2   398.4
   393.4   389.3   384.5   379.8     375   370.4   365.9   361.1   356.3   352.4
   347.6   342.8   338.8   334.8     331   327.7
Use DSS=False
CWMS InputPosition= 0
Use Fixed Start Time=False
Fixed Start Date/Time=07JUN1995,0000
Is Critical Boundary=False
Boundary Location=Main Gut        ,Downstream      ,0       ,        ,                ,                ,
Interval=1HOUR
Stage Hydrograph= 96
    .311    .358     .27    .073   -.187   -.451   -.659   -.759   -.716   -.534
   -.257    .052    .322    .478    .483    .346    .113   -.154    -.39   -.542
    -.57   -.458   -.239    .024    .264    .417    .431    .298    .051   -.243
   -.512     -.7   -.766   -.678    -.45   -.151    .145    .373    .475     .42
    .224    -.05    -.32   -.527   -.632   -.596   -.413   -.141    .141    .371
    .495     .47     .29    .008   -.293    -.54   -.695   -.718   -.585   -.331
   -.042    .212    .385    .426    .309    .066   -.221   -.468    -.63   -.677
   -.574   -.335   -.037    .237    .441    .532    .469    .256   -.035   -.314
   -.524   -.637   -.619   -.455   -.206    .043    .241    .353    .334    .167
   -.098   -.369   -.576   -.687   -.676   -.519
Use DSS=False
CWMS InputPosition= 0
Use Fixed Start Time=False
Fixed Start Date/Time=07JUN1995,0000
Is Critical Boundary=False

--- StephenvilleCrossi.u18 (unsteady flow) ---

Flow Title=Calibration Run, Dec 1986,mar1,11
Program Version=4.10
Use Restart= 0
Initial Flow Loc=Harrys River    ,Upstream        ,1826.936,22.6
Initial Flow Loc=Main Gut        ,Downstream      ,600     ,67.2
Initial Flow Loc=StGeorgesRiver  ,Upstream        ,1500    ,44.6
Initial Storage Elev=St. George's Riv,-0.44
Boundary Location=Harrys River    ,Upstream        ,1826.936,        ,                ,                ,
Interval=1HOUR
Flow Hydrograph= 428
    22.6    22.6    22.6    22.6    22.6    22.6    22.6    22.6    20.4    20.4
    20.4    20.4    20.4    20.4    20.4    20.4    20.4    20.4    20.4    20.4
    20.4    20.4    20.4    20.4    20.4    20.4    20.4    20.4    20.4    20.4
    20.4    20.4    26.3    26.3    26.3    26.3    26.3    26.3    26.3    26.3
    26.3    26.3    26.3    26.3    26.3    26.3    26.3    26.3    26.3    26.3
    26.3    26.3    26.3    26.3    26.3    26.3    31.5    31.5    31.5    31.5
    31.5    31.5    31.5    31.5    31.5    31.5    31.5    31.5    31.5    31.5
    31.5    31.5    31.5    31.5    31.5    31.5    31.5    31.5    31.5    31.5
    26.4    26.4    26.4    26.4    26.4    26.4    26.4    26.4    26.4    26.4
    26.4    26.4    26.4    26.4    26.4    26.4    26.4    26.4    26.4    26.4
    26.4    26.4    26.4    26.4      24      24      24      24      24      24
      24      24      24      24      24      24      24      24      24      24
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Use DSS=False
CWMS InputPosition= 0
Use Fixed Start Time=True
Fixed Start Date/Time=2dec1986,16:00
Is Critical Boundary=False
Boundary Location=StGeorgesRiver  ,Upstream        ,1500    ,        ,                ,                ,
Interval=1HOUR
Flow Hydrograph= 428
    44.6    44.6    44.6    44.6    44.6    44.6    44.6    44.6    40.2    40.2
    40.2    40.2    40.2    40.2    40.2    40.2    40.2    40.2    40.2    40.2
    40.2    40.2    40.2    40.2    40.2    40.2    40.2    40.2    40.2    40.2
    40.2    40.2    51.9    51.9    51.9    51.9    51.9    51.9    51.9    51.9
    51.9    51.9    51.9    51.9    51.9    51.9    51.9    51.9    51.9    51.9
    51.9    51.9    51.9    51.9    51.9    51.9    62.3    62.3    62.3    62.3
    62.3    62.3    62.3    62.3    62.3    62.3    62.3    62.3    62.3    62.3
    62.3    62.3    62.3    62.3    62.3    62.3    62.3    62.3    62.3    62.3
    52.1    52.1    52.1    52.1    52.1    52.1    52.1    52.1    52.1    52.1
    52.1    52.1    52.1    52.1    52.1    52.1    52.1    52.1    52.1    52.1
    52.1    52.1    52.1    52.1    47.3    47.3    47.3    47.3    47.3    47.3
    47.3    47.3    47.3    47.3    47.3    47.3    47.3    47.3    47.3    47.3
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Use DSS=False
CWMS InputPosition= 0
Use Fixed Start Time=True
Fixed Start Date/Time=2dec1986,16:00
Is Critical Boundary=False
Boundary Location=Main Gut        ,Downstream      ,0       ,        ,                ,                ,
Interval=1HOUR
Stage Hydrograph= 428
    -.44    -.49    -.46     -.3    -.19     .12     .25     .27     .13     -.1
    -.25    -.67    -.85     -.9     -.8    -.55    -.39     .13     .42     .53
     .61     .48     .37    -.04    -.29    -.39    -.49    -.41    -.32    -.01
     .17     .23     .23     .07    -.05    -.47    -.73    -.82    -.89    -.74
    -.62    -.14      .2     .34     .58     .56      .5     .17     -.1    -.22
    -.45    -.45    -.41    -.16     .05     .13     .26     .19     .11    -.25
    -.52    -.64    -.86    -.83    -.77    -.39    -.07     .08     .44     .53
     .53     .32     .09    -.03    -.33    -.42    -.42    -.28     -.1    -.01
      .2     .22     .19    -.05    -.29    -.41    -.72     -.8    -.79    -.58
    -.32    -.18     .22      .4     .44     .39     .24     .13    -.18    -.33
    -.37    -.35    -.24    -.16     .07     .17     .19      .1    -.07    -.18
    -.49    -.65    -.69    -.65     -.5    -.39    -.03     .18     .26     .36
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Use DSS=False
CWMS InputPosition= 0
Use Fixed Start Time=False
Fixed Start Date/Time=2dec1986,16:00
Is Critical Boundary=False

--- StephenvilleCrossi.u22 (unsteady flow) ---

Flow Title=Calibration-HighWater-Nov2010,Mar10,11
Program Version=4.10
Use Restart= 0
Initial Flow Loc=Harrys River    ,Upstream        ,1826.936,44.08
Initial Flow Loc=Main Gut        ,Downstream      ,600     ,131.16
Initial Flow Loc=StGeorgesRiver  ,Upstream        ,1500    ,87.08
Initial Storage Elev=St. George's Riv,0.28
Boundary Location=Harrys River    ,Upstream        ,1826.936,        ,                ,                ,
Interval=1HOUR
Flow Hydrograph= 93
   44.08    44.2   43.69   44.08   43.18   43.43   42.67   42.54   42.67   42.03
   42.41    41.9   41.51   41.38   41.51   41.38   41.38   41.38   40.74   40.49
   40.74   40.23   40.36   39.98   39.98   39.59   39.21   39.33   39.08   38.95
   38.95   38.95   38.44   38.31   38.31    37.8   38.18   38.69   38.05   38.05
   38.18   38.95   39.33   40.36   41.38   44.33   45.36   48.69   55.35   55.48
   54.71    54.2    52.4   51.51   51.12   49.71   49.07   48.56   48.56   47.92
   47.53   48.18   48.69   49.46   51.25   93.66   99.55   99.55   99.81   96.61
   93.79   88.92   86.61   86.36   88.92   88.53   89.05   87.51   87.13   85.46
   82.38   80.85   80.08   80.98   83.92   87.38   87.13   89.05   89.69   89.05
   87.51   86.36   84.82
Use DSS=False
CWMS InputPosition= 0
Use Fixed Start Time=True
Fixed Start Date/Time=03NOV2010,2000
Is Critical Boundary=False
Boundary Location=StGeorgesRiver  ,Upstream        ,1500    ,        ,                ,                ,
Interval=1HOUR
Flow Hydrograph= 93
   87.08   87.33   86.32   87.08    85.3   85.81   84.29   84.04   84.29   83.03
   83.78   82.77   82.01   81.76   82.01   81.76   81.76   81.76   80.49   79.99
   80.49   79.48   79.73   78.98   78.98   78.22   77.46   77.71    77.2   76.95
   76.95   76.95   75.94   75.68   75.68   74.67   75.43   76.44   75.18   75.18
   75.43   76.95   77.71   79.73   81.76   87.58   89.61   96.19  109.35   109.6
  108.08  107.07  103.53  101.76     101   98.21   96.95   95.93   95.93   94.67
   93.91   95.18   96.19   97.71  101.25  185.03  196.68  196.68  197.18  190.86
  185.29  175.67  171.11  170.61  175.67  174.91  175.92  172.88  172.13  168.83
  162.76  159.72   158.2  159.98   165.8  172.63  172.13  175.92  177.19  175.92
  172.88  170.61  167.57
Use DSS=False
CWMS InputPosition= 0
Use Fixed Start Time=True
Fixed Start Date/Time=03NOV2010,2000
Is Critical Boundary=False
Boundary Location=Main Gut        ,Downstream      ,0       ,        ,                ,                ,
Interval=1HOUR
Stage Hydrograph= 93
     .28     .17    -.02    -.26    -.47     -.6    -.62    -.53    -.33    -.08
     .17     .35     .42     .37      .2    -.03    -.28    -.48    -.58    -.56
    -.43    -.22     .01      .2     .29     .27     .13     -.1    -.36    -.57
     -.7    -.69    -.55    -.31    -.02     .25     .44      .5     .42     .23
    -.03     -.3     -.5    -.59    -.55     -.4    -.17     .06     .23      .3
     .24     .05     -.2    -.47    -.68    -.78    -.73    -.54    -.26     .06
     .34     .51     .55     .44     .22    -.06    -.32    -.51    -.58    -.51
    -.34    -.11     .11     .26     .28     .18    -.04    -.32    -.58    -.76
    -.82    -.72     -.5    -.18     .14     .41     .56     .56     .42     .18
     -.1    -.35    -.51
Use DSS=False
CWMS InputPosition= 0
Use Fixed Start Time=False
Is Critical Boundary=False

--- StephenvilleCrossi.u23 (unsteady flow) ---

Flow Title=Calibration-SurveyDate-Sep2010,Mar10,11
Program Version=4.10
Use Restart= 0
Initial Flow Loc=Harrys River    ,Upstream        ,1826.936,10.05
Initial Flow Loc=Main Gut        ,Downstream      ,600     ,29.9
Initial Flow Loc=StGeorgesRiver  ,Upstream        ,1500    ,19.85
Initial Storage Elev=St. George's Riv,0.076
Boundary Location=Harrys River    ,Upstream        ,1826.936,        ,                ,                ,
Interval=1HOUR
Flow Hydrograph= 96
   10.05   10.05   10.05   10.05   10.05   10.05   10.05   10.05   10.05   10.05
   10.05   10.05   10.05   10.05   10.05   10.05   10.05   10.05   10.05   10.05
   10.05   10.05   10.05   10.05    9.64    9.64    9.64    9.64    9.64    9.64
    9.64    9.64    9.64    9.64    9.64    9.64    9.64    9.64    9.64    9.64
    9.64    9.64    9.64    9.64    9.64    9.64    9.64    9.64    9.12    9.12
    9.12    9.12    9.12    9.12    9.12    9.12    9.12    9.12    9.12    9.12
    9.12    9.12    9.12    9.12    9.12    9.12    9.12    9.12    9.12    9.12
    9.12    9.12   11.76   11.76   11.76   11.76   11.76   11.76   11.76   11.76
   11.76   11.76   11.76   11.76   11.76   11.76   11.76   11.76   11.76   11.76
   11.76   11.76   11.76   11.76   11.76   11.76
Use DSS=False
CWMS InputPosition= 0
Use Fixed Start Time=False
Fixed Start Date/Time=03NOV2010,2000
Is Critical Boundary=False
Boundary Location=StGeorgesRiver  ,Upstream        ,1500    ,        ,                ,                ,
Interval=1HOUR
Flow Hydrograph= 96
   19.85   19.85   19.85   19.85   19.85   19.85   19.85   19.85   19.85   19.85
   19.85   19.85   19.85   19.85   19.85   19.85   19.85   19.85   19.85   19.85
   19.85   19.85   19.85   19.85   19.04   19.04   19.04   19.04   19.04   19.04
   19.04   19.04   19.04   19.04   19.04   19.04   19.04   19.04   19.04   19.04
   19.04   19.04   19.04   19.04   19.04   19.04   19.04   19.04   18.02   18.02
   18.02   18.02   18.02   18.02   18.02   18.02   18.02   18.02   18.02   18.02
   18.02   18.02   18.02   18.02   18.02   18.02   18.02   18.02   18.02   18.02
   18.02   18.02   23.24   23.24   23.24   23.24   23.24   23.24   23.24   23.24
   23.24   23.24   23.24   23.24   23.24   23.24   23.24   23.24   23.24   23.24
   23.24   23.24   23.24   23.24   23.24   23.24
Use DSS=False
CWMS InputPosition= 0
Use Fixed Start Time=False
Fixed Start Date/Time=03NOV2010,2000
Is Critical Boundary=False
Boundary Location=Main Gut        ,Downstream      ,0       ,        ,                ,                ,
Interval=1HOUR
Stage Hydrograph= 96
    .076    -.13   -.356   -.546   -.648   -.635   -.505   -.287   -.032    .201
    .357    .403    .331    .162   -.057   -.269   -.422   -.477   -.425   -.283
   -.095    .086    .206    .227    .138   -.043   -.274   -.497   -.657   -.709
   -.639   -.458   -.206     .06    .279    .405    .412    .305    .116   -.102
   -.294    -.41   -.426   -.341   -.184   -.003    .147    .219    .186    .049
   -.162     -.4   -.605   -.726    -.73   -.612   -.396   -.129    .131    .327
    .419    .394    .265    .071   -.134   -.297   -.378   -.361   -.257     -.1
    .061    .174    .202    .127    -.04   -.264   -.492    -.67   -.753   -.718
   -.569   -.336    -.07    .173    .342    .406     .36    .224    .038   -.145
    -.28   -.334   -.299    -.19   -.045    .091
Use DSS=False
CWMS InputPosition= 0
Use Fixed Start Time=False
Is Critical Boundary=False

--- StephenvilleCrossi.u24 (unsteady flow) ---

Flow Title=1:100, High Tide, -1hr offset
Program Version=4.10
Use Restart= 0
Initial Flow Loc=Harrys River    ,Upstream        ,1826.936,51.3
Initial Flow Loc=Main Gut        ,Downstream      ,600     ,152.6
Initial Flow Loc=StGeorgesRiver  ,Upstream        ,1500    ,101.3
Initial Storage Elev=St. George's Riv,-0.301
Boundary Location=Harrys River    ,Upstream        ,1826.936,        ,                ,                ,
Interval=1HOUR
Flow Hydrograph= 96
    51.3    51.2    51.1      51    50.9    50.9    50.8    50.7    50.6    50.5
    50.4    50.3    50.1      50    49.9    49.7    49.5    49.3    49.1    48.8
    48.6    48.4    48.1    48.2    48.3    48.4    48.4    49.4    49.9    50.2
    51.7    55.8    93.3   162.9   262.3   372.8   829.9   888.2   946.8   934.8
   844.8   782.5   724.7   668.3   612.6     613   612.3   611.4   610.4   621.5
   633.1   639.7   607.2   575.7   543.5   509.8     476   442.3   410.6   375.4
   354.7   335.8     319   306.1   292.4   280.8   267.1   257.9   251.5     245
   238.6   232.2     225   217.3   214.1   211.7   209.3   206.5   204.1   201.7
   199.2     197   194.6   192.2   189.8   187.5   185.2   182.8   180.4   178.4
     176   173.5   171.5   169.5   167.6   165.9
Use DSS=False
CWMS InputPosition= 0
Use Fixed Start Time=False
Fixed Start Date/Time=07JUN1995,0000
Is Critical Boundary=False
Boundary Location=StGeorgesRiver  ,Upstream        ,1500    ,        ,                ,                ,
Interval=1HOUR
Flow Hydrograph= 96
   101.3   101.1   100.9   100.8   100.6   100.5   100.3   100.2    99.9    99.7
    99.5    99.3      99    98.8    98.6    98.3    97.8    97.3      97    96.3
      96    95.7    95.1    95.2    95.4    95.6    95.7    97.6    98.6    99.2
   102.2   110.2   184.4   321.7   518.2   736.5  1639.6  1754.7  1870.6  1846.8
    1669    1546  1431.7  1320.2  1210.3  1211.1  1209.7  1207.9    1206  1227.8
  1250.8  1263.9  1199.6  1137.3  1073.8  1007.1   940.5   873.8   811.1   741.7
   700.8   663.5   630.1   604.7   577.8   554.7   527.8   509.5   496.8   484.1
   471.4   458.7   444.5   429.4     423   418.2   413.5   407.9   403.2   398.4
   393.4   389.3   384.5   379.8     375   370.4   365.9   361.1   356.3   352.4
   347.6   342.8   338.8   334.8     331   327.7
Use DSS=False
CWMS InputPosition= 0
Use Fixed Start Time=False
Fixed Start Date/Time=07JUN1995,0000
Is Critical Boundary=False
Boundary Location=Main Gut        ,Downstream      ,0       ,        ,                ,                ,
Interval=1HOUR
Stage Hydrograph= 96
   -.301   -.085    .143    .311    .358     .27    .073   -.187   -.451   -.659
   -.759   -.716   -.534   -.257    .052    .322    .478    .483    .346    .113
   -.154    -.39   -.542    -.57   -.458   -.239    .024    .264    .417    .431
    .298    .051   -.243   -.512     -.7   -.766   -.678    -.45   -.151    .145
    .373    .475     .42    .224    -.05    -.32   -.527   -.632   -.596   -.413
   -.141    .141    .371    .495     .47     .29    .008   -.293    -.54   -.695
   -.718   -.585   -.331   -.042    .212    .385    .426    .309    .066   -.221
   -.468    -.63   -.677   -.574   -.335   -.037    .237    .441    .532    .469
    .256   -.035   -.314   -.524   -.637   -.619   -.455   -.206    .043    .241
    .353    .334    .167   -.098   -.369   -.576
Use DSS=False
CWMS InputPosition= 0
Use Fixed Start Time=False
Fixed Start Date/Time=07JUN1995,0000
Is Critical Boundary=False

--- StephenvilleCrossi.u26 (unsteady flow) ---

Flow Title=1:100, High Tide, -3hr offset
Program Version=4.10
Use Restart= 0
Initial Flow Loc=Harrys River    ,Upstream        ,1826.936,51.3
Initial Flow Loc=Main Gut        ,Downstream      ,600     ,152.6
Initial Flow Loc=StGeorgesRiver  ,Upstream        ,1500    ,101.3
Initial Storage Elev=St. George's Riv,0.073
Boundary Location=Harrys River    ,Upstream        ,1826.936,        ,                ,                ,
Interval=1HOUR
Flow Hydrograph= 96
    51.3    51.2    51.1      51    50.9    50.9    50.8    50.7    50.6    50.5
    50.4    50.3    50.1      50    49.9    49.7    49.5    49.3    49.1    48.8
    48.6    48.4    48.1    48.2    48.3    48.4    48.4    49.4    49.9    50.2
    51.7    55.8    93.3   162.9   262.3   372.8   829.9   888.2   946.8   934.8
   844.8   782.5   724.7   668.3   612.6     613   612.3   611.4   610.4   621.5
   633.1   639.7   607.2   575.7   543.5   509.8     476   442.3   410.6   375.4
   354.7   335.8     319   306.1   292.4   280.8   267.1   257.9   251.5     245
   238.6   232.2     225   217.3   214.1   211.7   209.3   206.5   204.1   201.7
   199.2     197   194.6   192.2   189.8   187.5   185.2   182.8   180.4   178.4
     176   173.5   171.5   169.5   167.6   165.9
Use DSS=False
CWMS InputPosition= 0
Use Fixed Start Time=False
Fixed Start Date/Time=07JUN1995,0000
Is Critical Boundary=False
Boundary Location=StGeorgesRiver  ,Upstream        ,1500    ,        ,                ,                ,
Interval=1HOUR
Flow Hydrograph= 96
   101.3   101.1   100.9   100.8   100.6   100.5   100.3   100.2    99.9    99.7
    99.5    99.3      99    98.8    98.6    98.3    97.8    97.3      97    96.3
      96    95.7    95.1    95.2    95.4    95.6    95.7    97.6    98.6    99.2
   102.2   110.2   184.4   321.7   518.2   736.5  1639.6  1754.7  1870.6  1846.8
    1669    1546  1431.7  1320.2  1210.3  1211.1  1209.7  1207.9    1206  1227.8
  1250.8  1263.9  1199.6  1137.3  1073.8  1007.1   940.5   873.8   811.1   741.7
   700.8   663.5   630.1   604.7   577.8   554.7   527.8   509.5   496.8   484.1
   471.4   458.7   444.5   429.4     423   418.2   413.5   407.9   403.2   398.4
   393.4   389.3   384.5   379.8     375   370.4   365.9   361.1   356.3   352.4
   347.6   342.8   338.8   334.8     331   327.7
Use DSS=False
CWMS InputPosition= 0
Use Fixed Start Time=False
Fixed Start Date/Time=07JUN1995,0000
Is Critical Boundary=False
Boundary Location=Main Gut        ,Downstream      ,0       ,        ,                ,                ,
Interval=1HOUR
Stage Hydrograph= 96
    .073   -.187   -.451   -.659   -.759   -.716   -.534   -.257    .052    .322
    .478    .483    .346    .113   -.154    -.39   -.542    -.57   -.458   -.239
    .024    .264    .417    .431    .298    .051   -.243   -.512     -.7   -.766
   -.678    -.45   -.151    .145    .373    .475     .42    .224    -.05    -.32
   -.527   -.632   -.596   -.413   -.141    .141    .371    .495     .47     .29
    .008   -.293    -.54   -.695   -.718   -.585   -.331   -.042    .212    .385
    .426    .309    .066   -.221   -.468    -.63   -.677   -.574   -.335   -.037
    .237    .441    .532    .469    .256   -.035   -.314   -.524   -.637   -.619
   -.455   -.206    .043    .241    .353    .334    .167   -.098   -.369   -.576
   -.687   -.676   -.519   -.251     .04    .289
Use DSS=False
CWMS InputPosition= 0
Use Fixed Start Time=False
Fixed Start Date/Time=07JUN1995,0000
Is Critical Boundary=False

--- StephenvilleCrossi.u27 (unsteady flow) ---

Flow Title=1:100, High Tide, -4hr offset
Program Version=4.10
Use Restart= 0
Initial Flow Loc=Harrys River    ,Upstream        ,1826.936,51.3
Initial Flow Loc=Main Gut        ,Downstream      ,600     ,152.6
Initial Flow Loc=StGeorgesRiver  ,Upstream        ,1500    ,101.3
Initial Storage Elev=St. George's Riv,-0.187
Boundary Location=Harrys River    ,Upstream        ,1826.936,        ,                ,                ,
Interval=1HOUR
Flow Hydrograph= 96
    51.3    51.2    51.1      51    50.9    50.9    50.8    50.7    50.6    50.5
    50.4    50.3    50.1      50    49.9    49.7    49.5    49.3    49.1    48.8
    48.6    48.4    48.1    48.2    48.3    48.4    48.4    49.4    49.9    50.2
    51.7    55.8    93.3   162.9   262.3   372.8   829.9   888.2   946.8   934.8
   844.8   782.5   724.7   668.3   612.6     613   612.3   611.4   610.4   621.5
   633.1   639.7   607.2   575.7   543.5   509.8     476   442.3   410.6   375.4
   354.7   335.8     319   306.1   292.4   280.8   267.1   257.9   251.5     245
   238.6   232.2     225   217.3   214.1   211.7   209.3   206.5   204.1   201.7
   199.2     197   194.6   192.2   189.8   187.5   185.2   182.8   180.4   178.4
     176   173.5   171.5   169.5   167.6   165.9
Use DSS=False
CWMS InputPosition= 0
Use Fixed Start Time=False
Fixed Start Date/Time=07JUN1995,0000
Is Critical Boundary=False
Boundary Location=StGeorgesRiver  ,Upstream        ,1500    ,        ,                ,                ,
Interval=1HOUR
Flow Hydrograph= 96
   101.3   101.1   100.9   100.8   100.6   100.5   100.3   100.2    99.9    99.7
    99.5    99.3      99    98.8    98.6    98.3    97.8    97.3      97    96.3
      96    95.7    95.1    95.2    95.4    95.6    95.7    97.6    98.6    99.2
   102.2   110.2   184.4   321.7   518.2   736.5  1639.6  1754.7  1870.6  1846.8
    1669    1546  1431.7  1320.2  1210.3  1211.1  1209.7  1207.9    1206  1227.8
  1250.8  1263.9  1199.6  1137.3  1073.8  1007.1   940.5   873.8   811.1   741.7
   700.8   663.5   630.1   604.7   577.8   554.7   527.8   509.5   496.8   484.1
   471.4   458.7   444.5   429.4     423   418.2   413.5   407.9   403.2   398.4
   393.4   389.3   384.5   379.8     375   370.4   365.9   361.1   356.3   352.4
   347.6   342.8   338.8   334.8     331   327.7
Use DSS=False
CWMS InputPosition= 0
Use Fixed Start Time=False
Fixed Start Date/Time=07JUN1995,0000
Is Critical Boundary=False
Boundary Location=Main Gut        ,Downstream      ,0       ,        ,                ,                ,
Interval=1HOUR
Stage Hydrograph= 96
   -.187   -.451   -.659   -.759   -.716   -.534   -.257    .052    .322    .478
    .483    .346    .113   -.154    -.39   -.542    -.57   -.458   -.239    .024
    .264    .417    .431    .298    .051   -.243   -.512     -.7   -.766   -.678
    -.45   -.151    .145    .373    .475     .42    .224    -.05    -.32   -.527
   -.632   -.596   -.413   -.141    .141    .371    .495     .47     .29    .008
   -.293    -.54   -.695   -.718   -.585   -.331   -.042    .212    .385    .426
    .309    .066   -.221   -.468    -.63   -.677   -.574   -.335   -.037    .237
    .441    .532    .469    .256   -.035   -.314   -.524   -.637   -.619   -.455
   -.206    .043    .241    .353    .334    .167   -.098   -.369   -.576   -.687
   -.676   -.519   -.251     .04    .289    .465
Use DSS=False
CWMS InputPosition= 0
Use Fixed Start Time=False
Fixed Start Date/Time=07JUN1995,0000
Is Critical Boundary=False

--- StephenvilleCrossi.u28 (unsteady flow) ---

Flow Title=1:100, Neap Tide, -1hr offset
Program Version=4.10
Use Restart= 0
Initial Flow Loc=Harrys River    ,Upstream        ,1826.936,51.3
Initial Flow Loc=Main Gut        ,Downstream      ,600     ,152.6
Initial Flow Loc=StGeorgesRiver  ,Upstream        ,1500    ,101.3
Initial Storage Elev=St. George's Riv,0.154
Boundary Location=Harrys River    ,Upstream        ,1826.936,        ,                ,                ,
Interval=1HOUR
Flow Hydrograph= 96
    51.3    51.2    51.1      51    50.9    50.9    50.8    50.7    50.6    50.5
    50.4    50.3    50.1      50    49.9    49.7    49.5    49.3    49.1    48.8
    48.6    48.4    48.1    48.2    48.3    48.4    48.4    49.4    49.9    50.2
    51.7    55.8    93.3   162.9   262.3   372.8   829.9   888.2   946.8   934.8
   844.8   782.5   724.7   668.3   612.6     613   612.3   611.4   610.4   621.5
   633.1   639.7   607.2   575.7   543.5   509.8     476   442.3   410.6   375.4
   354.7   335.8     319   306.1   292.4   280.8   267.1   257.9   251.5     245
   238.6   232.2     225   217.3   214.1   211.7   209.3   206.5   204.1   201.7
   199.2     197   194.6   192.2   189.8   187.5   185.2   182.8   180.4   178.4
     176   173.5   171.5   169.5   167.6   165.9
Use DSS=False
CWMS InputPosition= 0
Use Fixed Start Time=False
Fixed Start Date/Time=07JUN1995,0000
Is Critical Boundary=False
Boundary Location=StGeorgesRiver  ,Upstream        ,1500    ,        ,                ,                ,
Interval=1HOUR
Flow Hydrograph= 96
   101.3   101.1   100.9   100.8   100.6   100.5   100.3   100.2    99.9    99.7
    99.5    99.3      99    98.8    98.6    98.3    97.8    97.3      97    96.3
      96    95.7    95.1    95.2    95.4    95.6    95.7    97.6    98.6    99.2
   102.2   110.2   184.4   321.7   518.2   736.5  1639.6  1754.7  1870.6  1846.8
    1669    1546  1431.7  1320.2  1210.3  1211.1  1209.7  1207.9    1206  1227.8
  1250.8  1263.9  1199.6  1137.3  1073.8  1007.1   940.5   873.8   811.1   741.7
   700.8   663.5   630.1   604.7   577.8   554.7   527.8   509.5   496.8   484.1
   471.4   458.7   444.5   429.4     423   418.2   413.5   407.9   403.2   398.4
   393.4   389.3   384.5   379.8     375   370.4   365.9   361.1   356.3   352.4
   347.6   342.8   338.8   334.8     331   327.7
Use DSS=False
CWMS InputPosition= 0
Use Fixed Start Time=False
Fixed Start Date/Time=07JUN1995,0000
Is Critical Boundary=False
Boundary Location=Main Gut        ,Downstream      ,0       ,        ,                ,                ,
Interval=1HOUR
Stage Hydrograph= 96
    .154    .092   -.045   -.193    -.31   -.394   -.436   -.405   -.292   -.127
     .05    .206    .305    .309    .207    .048   -.105   -.234   -.333   -.372
   -.326   -.211   -.064    .081    .193    .231    .169    .031   -.122   -.255
   -.361   -.418    -.39   -.279   -.115    .061    .209    .289    .266    .142
   -.029   -.192   -.329   -.421   -.435   -.355   -.205   -.022    .151    .273
    .305    .232    .084   -.082   -.233    -.35   -.403   -.366   -.247   -.079
    .093     .22    .265    .207    .058   -.128   -.301   -.433   -.499   -.473
   -.352   -.161    .055    .241    .352    .364    .271    .105   -.078   -.237
   -.347   -.381   -.326   -.193   -.021    .135    .223    .223    .128   -.047
   -.248   -.419   -.526   -.549   -.474   -.306
Use DSS=False
CWMS InputPosition= 0
Use Fixed Start Time=False
Fixed Start Date/Time=07JUN1995,0000
Is Critical Boundary=False

--- StephenvilleCrossi.g11 (geometry) ---

Geom Title=StephenvilleX, Section10- Mar9,2011
Program Version=4.10
